--- INDIANCK.prj (project) ---

Proj Title=INDIANCK
Current Plan=p01
Default Exp/Contr=0,0
English Units
Geom File=g01
Flow File=f01
Plan File=p01
Background Map Layer=Final_Streamlines
Background Map Layer=QC
BEGIN DESCRIPTION:
Stream Name: Indian Creek
Flood Zone: Approximate
Summers County, West Virginia
HEC-RAS Version: 5.0.7
Hydrology Method:
Regression.
Model Notes:
END DESCRIPTION:
DSS Export Rating Curves= 0
DSS Export Rating Curve Sorted= 0
DSS Export Volume Flow Curves= 0
DXF OffsetX= 0
DXF OffsetY= 0
DXF ScaleX= 0
DXF ScaleY= 0

--- INDIANCK.p01 (plan) ---

Plan Title=Floodplain
Program Version=5.07
Short Identifier=Floodplain
Geom File=g01
Flow File=f01
Subcritical Flow
K Sum by GR= 0
Std Step Tol= 0.01
Critical Tol= 0.01
Num of Std Step Trials= 20
Max Error Tol= 0.3
Flow Tol Ratio= 0.001
Split Flow NTrial= 30
Split Flow Tol= 0.02
Split Flow Ratio= 0.02
Log Output Level= 0
Friction Slope Method= 1
Unsteady Friction Slope Method= 2
Unsteady Bridges Friction Slope Method= 1
Parabolic Critical Depth
Global Vel Dist= 0 , 0 , 0
Global Log Level= 0
CheckData=True
Encroach Param=-1 ,0,0, 0
Mapping Interval=1HOUR
Computation Time Step Use Courant=        0
Computation Time Step Use Time Series=    0
Computation Time Step Count To Double=0
Computation Time Step Max Doubling=0
Computation Time Step Max Halving=0
Computation Time Step Residence Courant=0
Run HTab= 0
Run UNet= 0
Run Sediment= 0
Run PostProcess= 0
Run WQNet= 0
Run RASMapper= 0
UNET Theta= 0
UNET Theta Warmup= 0
UNET ZTol= 0
UNET ZSATol= 0
UNET MxIter= 0
UNET Max Iter WO Improvement= 0
UNET MaxInSteps= 0
UNET DtIC= 0
UNET DtMin= 0
UNET MaxCRTS= 0
UNET WFStab= 0
UNET SFStab= 0
UNET WFX= 1
UNET SFX= 1
UNET 1D Methodology=Finite Difference
UNET DSS MLevel= 1
UNET Pardiso=0
UNET DZMax Abort= 0
UNET Use Existing IB Tables= 0
UNET Froude Reduction=False
UNET Froude Limit= 0
UNET Froude Power= 0
UNET D1 Cores= 0
UNET D2 Coriolis=0
UNET D2 Cores= 0
UNET D2 Theta= 1
UNET D2 Theta Warmup= 1
UNET D2 Z Tol= 0.01
UNET D2 Volume Tol= 0.01
UNET D2 Max Iterations= 20
UNET D2 Equation= 0
UNET D2 RampUpFraction=0.1
UNET D2 TimeSlices= 1
UNET D2 BCVolumeCheck=0
UNET D1D2 MaxIter= 0
UNET D1D2 ZTol=0.01
UNET D1D2 QTol=0.1
UNET D1D2 MinQTol=1
Write IC File= 0
Write IC File at Fixed DateTime=0
Write IC File at Sim End=0
Echo Input=False
Echo Parameters=False
Echo Output=False
Write Detailed= 0
HDF Write Warmup=0
HDF Write Time Slices=0
HDF Flush=0
HDF Face Node Velocities=0
HDF Compression= 1
HDF Chunk Size= 1
HDF Spatial Parts= 1
HDF Use Max Rows=0
HDF Fixed Rows= 1
Calibration Method= 0
Calibration Iterations= 20
Calibration Max Change=0.05
Calibration Tolerance=0.2
Calibration Maximum=1.5
Calibration Minimum=0.5
Calibration Optimization Method= 1
WQ AD Non Conservative
WQ ULTIMATE=-1
WQ Max Comp Step=1HOUR
WQ Output Interval=15MIN
WQ Output Selected Increments= 0
WQ Output face flow=0
WQ Output face velocity=0
WQ Output face area=0
WQ Output face dispersion=0
WQ Output cell volume=0
WQ Output cell surface area=0
WQ Output cell continuity=0
WQ Output cumulative cell continuity=0
WQ Output face conc=0
WQ Output face dconc_dx=0
WQ Output face courant=0
WQ Output face peclet=0
WQ Output face adv mass=0
WQ Output face disp mass=0
WQ Output cell mass=0
WQ Output cell source sink temp=0
WQ Output nsm pathways=0
WQ Output nsm derived pathways=0
WQ Output MaxMinRange=-1
WQ Daily Max Min Mean=-1
WQ Daily Range=0
WQ Daily Time=0
WQ Create Restart=0
WQ Fixed Restart=0
WQ System Summary=0
WQ Write To DSS=0
WQ Use Fixed Temperature=0
Sorting and Armoring Iterations= 10
XS Update Threshold= 0.02
Bed Roughness Predictor= 0
Hydraulics Update Threshold= 0.02
Energy Slope Method= 1
Volume Change Method= 1
Sediment Retention Method= 0
XS Weighting Method= 0
Number of US Weighted Cross Sections= 1
Number of DS Weighted Cross Sections= 1
Upstream XS Weight=0
Main XS Weight=1
Downstream XS Weight=0
Number of DS XS's Weighted with US Boundary= 1
Upstream Boundary Weight= 1
Weight of XSs Associated with US Boundary= 0
Number of US XS's Weighted with DS Boundary= 1
Downstream Boundary Weight= 0.5
Weight of XSs Associated with DS Boundary= 0.5
Percentile Method= 0
Sediment Output Level= 3
Mass or Volume Output= 0
Output Increment Type= 1
Profile and TS Output Increment= 1
XS Output Flag= 0
XS Output Increment= 10
Write Gradation File= 0
Read Gradation Hotstart= 0
Write HDF5 File= 1
Write Binary Output= 1
Write DSS Sediment File= 0
SV Curve= 0
Specific Gage Flag= 0

--- INDIANCK.f01 (steady flow) ---

Flow Title=Flows
Program Version=5.07
Number of Profiles= 6
Profile Names=01pct,10pct,04pct,02pct,0_2pct,01plus
River Rch & RM=INDIANCK,Main            ,30858
   17921   10822   13493   15636   23468   26506
River Rch & RM=INDIANCK,Main            ,20476
   20007   12133   15096   17473   26146   29591
Boundary for River Rch & Prof#=INDIANCK,Main            , 1
Up Type= 0
Dn Type= 3
Dn Slope=0.00393
Boundary for River Rch & Prof#=INDIANCK,Main            , 2
Up Type= 0
Dn Type= 3
Dn Slope=0.00393
Boundary for River Rch & Prof#=INDIANCK,Main            , 3
Up Type= 0
Dn Type= 3
Dn Slope=0.00393
Boundary for River Rch & Prof#=INDIANCK,Main            , 4
Up Type= 0
Dn Type= 3
Dn Slope=0.00393
Boundary for River Rch & Prof#=INDIANCK,Main            , 5
Up Type= 0
Dn Type= 3
Dn Slope=0.00393
Boundary for River Rch & Prof#=INDIANCK,Main            , 6
Up Type= 0
Dn Type= 3
Dn Slope=0.00393
DSS Import GetInterval= 0
DSS Import GetPeak= 0
DSS Import FillOption= 0

--- INDIANCK.g01 (geometry) ---

Geom Title=Geometry
Program Version=5.07

River Reach=INDIANCK        ,Main
Reach XY= 30
2028446.86736687189471.9306230822028004.98100002189549.036999988
2027695.73599999 189904.940000022027454.85100001190759.974999997
2026515.84500003192636.1060000362025011.93900001193261.106000047
2024460.53100001193140.118999988     2024326.175192232.460000022
2023379.99400001191120.0469999972023065.75800002189573.171999993
2022771.48800001189424.7350000342022412.11299999 189502.86000004
2022190.75800002 189984.63100003     2021159.508190745.046999985
     2020242.842      192071.4362020708.22700002193840.006000027
     2020313.445194032.7050000252019947.51600001193831.981000024
     2019572.133193024.0139999942018811.70900002192496.246000029
2017250.94500001192256.6629999972017334.27900001      191626.454
     2017737.056 191397.287999992018459.27900001191338.260000037
2018813.44500003190728.885000014     2018323.862 189918.12100001
2016153.72299999187475.413000014     2015413.089187485.839000022
     2013541.932188469.5020000332012671.12400002188659.822999993

Type RM Length L Ch R = 1 ,30858   ,158.7,156,153
XS GIS Cut Line= 3
     2027797.084      189124.128     2028573.126      190191.837
     2028600.209      190684.574
#Sta/Elev= 30
       0 1815.92    42.6 1781.87    68.8 1764.88   117.9  1727.7   176.9 1698.38
     285 1629.54   304.6 1614.59   337.4 1584.56     357 1561.84     393 1531.19
     416 1508.35   422.5 1504.57   435.6 1502.55   442.2 1499.11   455.3 1498.63
   501.1 1498.74   517.5 1501.04   550.2 1501.84   579.7 1509.07  1195.5 1512.83
  1257.7 1520.66  1316.7 1533.56  1359.2  1534.9  1391.8 1544.41  1571.6 1557.82
  1617.3 1558.74  1633.7 1562.35    1686 1565.36  1774.2    1581  1813.4 1590.14
#Mann= 6 ,-1 , 0
       0      .1       0   435.6    .045       0   517.5      .1       0
     640    .035       0    1260     .04       0 1459.94      .1       0
#XS Ineff= 2 , 0
                         1083.09         1542.98
Permanent Ineff=
       F       F
Bank Sta=435.6,517.5
XS Rating Curve= 0 ,0
Exp/Cntr(USF)=0,0
Exp/Cntr=0.3,0.1

Type RM Length L Ch R = 1 ,30702   ,505,510.6,506.1
XS GIS Cut Line= 3
     2027645.348       189226.24     2028468.265       190226.24
     2028516.876      190618.602
#Sta/Elev= 30
       0 1887.73    19.7 1877.16    45.9 1857.45    91.8 1818.77   111.5 1799.96
   183.6 1743.23   236.1 1694.28   252.5 1668.14   278.7 1637.71     377  1542.5
   396.7 1525.77   419.7 1509.14   439.3 1499.89   491.6 1498.76   508.2 1499.03
     518 1501.66   550.8 1501.05   560.6 1506.96   570.5 1509.28   626.2 1508.48
   711.5  1511.1  1042.6 1510.34  1124.6 1512.46  1213.1 1519.03  1295.1 1529.42
  1409.4 1540.34  1523.8 1545.36  1585.9  1550.9  1638.2 1560.66  1690.4 1567.23
#Mann= 5 ,-1 , 0
       0      .1       0   439.3    .045       0     518      .1       0
     630    .035       0 1295.06     .04       0
#XS Ineff= 2 , 0
                         1041.83         1554.61
Permanent Ineff=
       F       F
Bank Sta=439.3,518
XS Rating Curve= 0 ,0
Exp/Cntr(USF)=0,0
Exp/Cntr=0.3,0.1

Type RM Length L Ch R = 1 ,30191   ,443,408.5,415.3
XS GIS Cut Line= 3
     2027312.015      189615.129     2028136.897       190551.31
     2028360.626      190691.518
#Sta/Elev= 30
       0 1879.23      59 1830.02   137.6 1756.52   173.6 1729.78   216.1 1690.76
   232.5 1678.47   248.9 1660.85   258.7 1647.02   307.8 1593.84   317.7  1580.3
   340.6 1559.56   363.5  1542.4   389.7 1531.36   425.7 1508.55   435.6 1504.92
   455.2 1501.76   468.3 1497.95   530.5 1498.21   546.9 1501.13   569.8 1504.14
   586.2 1509.13   668.1  1507.7   740.1 1508.88   789.3 1506.95   867.8 1508.24
  1106.9 1513.55  1247.7 1520.24  1387.9 1530.34  1498.7 1549.58  1511.8 1550.06
#Mann= 6 ,-1 , 0
       0     .12       0      30      .1       0   455.2    .045       0
   546.9      .1       0     670    .035       0 1377.74     .04       0
#XS Ineff= 2 , 0
                           976.5         1542.54
Permanent Ineff=
       F       F
Bank Sta=455.2,546.9
XS Rating Curve= 0 ,0
Exp/Cntr(USF)=0,0
Exp/Cntr=0.3,0.1

Type RM Length L Ch R = 1 ,29783   ,353.6,352.2,337.7
XS GIS Cut Line= 4
     2027131.459      190160.268     2027423.126      190306.102
     2028107.153      190792.213     2028204.376      190896.379
#Sta/Elev= 30
       0 1831.38     9.8 1819.81    29.4  1803.1    55.4 1778.52   110.9 1731.07
   156.5 1686.01     163 1677.76   176.1 1667.71   189.1 1653.27   198.9 1645.92
   247.8 1602.02     313 1548.25   342.5 1528.46   362.2 1519.39   414.6    1512
   450.7 1499.81   460.5 1497.97   522.8 1497.84   535.9 1498.06   542.4 1501.07
   552.3 1505.46   565.4 1506.55   650.6 1507.58   742.4 1512.08   935.8 1515.63
  1106.2 1523.47  1165.3  1529.3  1275.4 1545.73  1294.8 1545.54  1307.8 1549.24
#Mann= 5 ,-1 , 0
       0      .1       0   450.7    .045       0   542.4      .1       0
  606.09    .035       0 1225.26     .04       0
#XS Ineff= 2 , 0
                          854.44         1542.98
Permanent Ineff=
       F       F
Bank Sta=450.7,542.4
XS Rating Curve= 0 ,0
Exp/Cntr(USF)=0,0
Exp/Cntr=0.3,0.1

Type RM Length L Ch R = 1 ,29431   ,362.7,365.6,367.1
XS GIS Cut Line= 3
     2027002.302      190475.484     2027867.872      190961.513
     2028034.922      191167.969
#Sta/Elev= 30
       0 1778.21    32.8 1773.66    68.8 1765.79    88.5 1759.12   108.1 1748.98
   163.8 1710.33     190 1683.41   229.3 1652.53     285    1601     308 1581.95
   317.8 1570.92   353.8  1544.7   399.7 1519.24   419.4 1511.17   484.9 1500.58
   491.4 1498.16   560.2  1497.8   563.5  1497.9   570.1  1502.3   579.9 1505.03
   874.8 1515.18     970 1522.61  1038.6 1529.88  1068.1 1536.53    1091 1538.53
  1100.9 1545.33  1123.8 1554.71  1205.8 1597.28  1235.3 1608.94  1258.3 1615.44
#Mann= 6 ,-1 , 0
       0      .1       0   484.9    .045       0   570.1      .1       0
     700    .035       0     970     .04       0 1122.69      .1       0
#XS Ineff= 2 , 0
                          780.23         1545.94
Permanent Ineff=
       F       F
Bank Sta=484.9,570.1
XS Rating Curve= 0 ,0
Exp/Cntr(USF)=0,0
Exp/Cntr=0.3,0.1

Type RM Length L Ch R = 1 ,29065   ,465.7,466.4,470.3
XS GIS Cut Line= 4
2026826.91321725190786.8782762232027181.89736212190987.421267156
2027587.59352769191234.0660950842027804.27216157 191400.03270827
#Sta/Elev= 30
       0 1667.07   154.2 1663.43   217.3 1657.49   239.2 1653.82   263.2  1647.4
   280.1  1640.8   298.5 1630.74   359.6 1588.91   411.6 1547.47   446.1 1523.74
   470.8 1510.61   510.4 1501.06   515.2 1498.12   519.1 1497.74   595.9 1497.94
   601.1 1501.35   607.4 1504.67   638.1 1504.81   701.6 1508.47   726.4 1512.12
   751.6 1513.41   775.4 1524.01   777.8 1527.93     784 1542.79   787.8 1546.95
   862.4 1570.94   903.9 1580.47   995.5 1595.61  1102.7 1605.85 1155.44  1609.2
#Mann= 5 ,-1 , 0
       0      .1       0   510.4    .045       0   601.1      .1       0
  647.71     .04       0  847.71      .1       0
Bank Sta=510.4,601.1
XS Rating Curve= 0 ,0
Exp/Cntr(USF)=0,0
Exp/Cntr=0.3,0.1

Type RM Length L Ch R = 1 ,28599   ,590.4,594.1,594.8
XS GIS Cut Line= 4
2026739.28642611191242.403166922 2026886.9474745191343.081154461
2027350.06621718191645.1151170792027564.84592393 191792.77616547
#Sta/Elev= 30
       0 1600.59    66.6 1590.19    94.8 1583.25   130.7 1572.39   142.1 1566.84
   209.7 1539.44   248.8 1528.88   331.1 1511.01   370.3 1507.21   393.3 1503.56
   401.6 1498.35     476 1497.72   479.9 1497.91   487.8 1503.52   490.5 1504.21
   515.2 1503.89   573.4 1506.97     621  1506.5     664 1507.56   680.7 1510.01
   695.4 1510.06   707.1 1519.93   726.7 1530.65   770.4 1558.17   786.5 1566.27
   818.2 1578.33   842.1 1584.22   878.5 1589.76   925.7 1594.18   992.3 1596.97
#Mann= 7 ,-1 , 0
       0      .1       0   393.3    .045       0   490.5      .1       0
  628.72     .04       0  741.62      .1       0  861.62     .08       0
  981.62      .1       0
Bank Sta=393.3,490.5
XS Rating Curve= 0 ,0
Exp/Cntr(USF)=0,0
Exp/Cntr=0.3,0.1

Type RM Length L Ch R = 1 ,28004   ,433.3,431.5,432.6
XS GIS Cut Line= 4
2026511.08298769191765.9287021262026652.03217024191880.030421337
2027108.43904709192208.9118472982027323.21875384192383.420359033
#Sta/Elev= 30
       0  1585.7    66.2 1587.75   114.7 1587.47     145 1584.58     166 1580.72
   179.3 1576.81   191.8 1571.68   260.2 1535.28   285.8 1524.85   349.2 1501.76
   357.3 1497.17   361.3 1496.35   412.7 1497.28   433.5    1501   482.6 1505.77
   645.4 1508.66   657.9 1509.48   666.5 1512.03     683 1512.55     686 1513.65
   708.8 1528.61   717.2 1537.32   732.3 1547.53   751.1 1557.35   778.7  1563.8
   832.7 1573.76   868.2 1581.62   910.4  1592.7   956.3 1607.23  1020.6 1622.59
#Mann= 5 ,-1 , 0
       0      .1       0   349.2    .045       0   433.5      .1       0
  571.34     .04       0  721.34      .1       0
Bank Sta=349.2,433.5
XS Rating Curve= 0 ,0
Exp/Cntr(USF)=0,0
Exp/Cntr=0.3,0.1

Type RM Length L Ch R = 1 ,27573   ,487.7,503,517.5
XS GIS Cut Line= 4
2026282.87954927192121.657591431  2026457.388061192262.606773986
2026880.23560867192557.9288707672027182.26957128192665.318724142
#Sta/Elev= 30
       0 1570.15   140.7 1571.32   184.2  1570.9   243.7 1569.18   259.7 1567.13
     272 1564.39   283.7 1559.93   295.4  1553.6   344.8 1522.94   367.7 1511.67
   390.4 1506.78   406.1  1505.2   427.3 1500.91   431.8 1499.55   436.7 1496.83
   439.8 1496.26   499.8 1496.23   509.9 1499.63   515.8 1500.26   535.5 1504.58
   569.9 1505.16   579.8 1506.25   601.7 1505.64   611.8 1507.08   627.6 1512.33
   667.6 1529.52   718.9 1544.71   807.5 1563.92   951.4 1593.08  1060.6 1617.19
#Mann= 5 ,-1 , 0
       0     .12       0     120      .1       0   427.3    .045       0
   515.8     .04       0  724.32      .1       0
Bank Sta=427.3,515.8
XS Rating Curve= 0 ,0
Exp/Cntr(USF)=0,0
Exp/Cntr=0.3,0.1

Type RM Length L Ch R = 1 ,27070   ,500.1,525.1,536.5
XS GIS Cut Line= 4
2025974.13372081192396.8440907052026162.06596422192571.352602439
2026464.09992684192927.0814917442026652.03217024 193148.57306433
#Sta/Elev= 30
       0 1559.28    98.7 1556.02   199.6 1555.68   252.7    1553   291.2  1546.1
   321.8 1538.89   331.1 1535.27   368.3 1515.55   391.6 1508.05   420.9 1503.64
   433.1 1499.57   459.1 1501.32   470.7 1500.75   481.2 1496.35     494 1495.81
   554.3 1496.19   561.5 1500.02   570.8 1504.29   610.3 1510.79   640.4 1518.96
   661.2 1520.69   686.6 1525.79   752.3 1549.56   803.6 1564.07   822.2 1570.96
   838.4 1570.41   848.8 1577.47   881.4 1586.67   992.1 1622.27  1013.6 1627.08
#Mann= 6 ,-1 , 0
       0     .12       0  276.46      .1       0   470.7    .045       0
   561.5      .1       0  586.46     .04       0  666.46      .1       0
Bank Sta=470.7,561.5
XS Rating Curve= 0 ,0
Exp/Cntr(USF)=0,0
Exp/Cntr=0.3,0.1

Type RM Length L Ch R = 1 ,26545   ,577.2,595.7,617
XS GIS Cut Line= 4
2025678.81162403192537.7932732592025759.35401406192705.589919158
2025974.13372081 193215.69172269 2026101.6591717193376.776502753
#Sta/Elev= 30
       0 1544.95    52.5 1537.69     129    1532   171.1 1527.78   216.5 1521.31
   290.4 1512.96   379.4 1508.22   388.8 1505.74   393.6 1499.68   397.2 1496.44
   411.3 1494.31   463.9 1494.73   496.9 1499.52   507.6 1500.57   539.6 1500.84
   557.4  1503.6   596.6  1504.8   610.8 1508.91   621.5 1515.76   636.8  1516.5
   639.3 1518.09   646.4 1525.41   682.3 1549.85   731.8 1580.82     789 1613.13
   830.6 1631.43   844.6 1639.57   863.3 1641.64     883  1650.2   945.1 1668.03
#Mann= 5 ,-1 , 0
       0      .1       0   393.6    .045       0   496.9      .1       0
  596.13     .04       0  706.13      .1       0
#XS Ineff= 2 , 0
          383.23 1523.04
Permanent Ineff=
       F       F
Bank Sta=393.6,496.9
XS Rating Curve= 0 ,0
Exp/Cntr(USF)=0,0
Exp/Cntr=0.3,0.1

Type RM Length L Ch R = 1 ,25949   ,1088.9,1215.7,1333.4
XS GIS Cut Line= 4
2025282.81153971192356.5728956892025255.96407637192712.301784994
2025356.64206391193423.759563604 2025430.4725881193826.471513761
#Sta/Elev= 30
       0 1543.76    77.9 1532.15   216.1 1518.28   417.2  1510.3   619.3 1507.15
   726.2 1503.19   781.7 1503.07  793.881500.474   804.9 1499.18   814.8 1495.09
   894.4 1493.81  915.741500.474   934.1 1511.98   950.7 1511.99   960.6 1520.77
  1002.2 1544.31  1083.3  1595.3    1130 1626.55    1150 1642.45  1163.3 1644.79
  1173.2 1651.24  1183.3 1659.76  1226.7 1683.61  1236.7 1685.62  1263.4 1702.03
  1286.7 1713.36  1333.4  1731.3  1383.5 1743.68  1416.8 1749.12  1484.7 1757.31
#Mann= 5 ,-1 , 0
       0      .1       0  793.88    .045       0  915.74      .1       0
  936.74     .04       0 1026.74      .1       0
#XS Ineff= 2 , 0
           601.2 1538.35
Permanent Ineff=
       F       F
Bank Sta=793.88,915.74
XS Rating Curve= 0 ,0
Exp/Cntr(USF)=0,0
Exp/Cntr=0.3,0.1

Type RM Length L Ch R = 1 ,24734   ,704,711.1,680
XS GIS Cut Line= 4
 2025262.6759422192316.3017006732024920.37078457192651.894992471
 2024141.7943476192913.6577600722023866.60784833193074.742540135
#Sta/Elev= 30
       0    1542   150.7 1523.98   345.6 1509.77   613.3 1505.56   665.2 1506.83
     723 1503.21   765.6 1506.39   775.9 1502.12   789.8 1507.66   807.1 1505.28
     859 1504.82  939.771496.981   990.6 1491.37  1028.6 1490.88  1080.5 1491.04
 1116.561496.982  1149.8 1503.49  1170.5 1518.68  1191.3 1528.46  1205.1 1538.31
    1219 1540.61  1267.4 1588.78  1288.5 1604.33  1295.1 1611.97  1302.2 1623.89
  1416.2 1703.98  1440.4 1719.47  1473.3 1735.92  1575.9 1797.43  1619.6 1818.95
#Mann= 7 ,-1 , 0
       0      .1       0  939.77    .045       0 1116.56      .1       0
 1139.37     .08       0 1209.37     .04       0 1239.37      .1       0
 1350.77     .08       0
#XS Ineff= 2 , 0
           693.7 1535.96
Permanent Ineff=
       F       F
Bank Sta=939.77,1116.56
XS Rating Curve= 0 ,0
Exp/Cntr(USF)=0,0
Exp/Cntr=0.3,0.1

Type RM Length L Ch R = 1 ,24022   ,692.8,692,680
XS GIS Cut Line= 4
2024920.37078457191906.8778846812024578.06562694192014.267738056
2023786.06545829192369.9966273612023537.72642237192490.810212408
#Sta/Elev= 30
       0 1611.28    36.7 1613.08   122.7 1598.02   208.7 1592.42   381.6 1568.37
   528.4 1551.72   548.3 1546.52   622.7 1508.05   657.5 1494.16   672.9 1487.58
   698.1  1487.5   712.5 1488.03   727.2 1493.71   773.6  1488.3   813.2 1488.24
   841.9 1494.27   867.1 1498.97   946.2 1503.52    1029 1511.89  1068.5 1518.75
  1094.3 1527.53  1147.7 1551.84  1171.2 1565.41  1188.6  1567.1  1201.6 1577.65
  1263.3 1611.61  1369.1 1674.17  1429.5 1715.15  1456.6    1730  1503.1 1764.64
#Mann= 5 ,-1 , 0
       0      .1       0   657.5    .045       0   841.9      .1       0
 1098.76     .04       0 1208.76     .08       0
Bank Sta=657.5,841.9
XS Rating Curve= 0 ,0
Exp/Cntr(USF)=0,0
Exp/Cntr=0.3,0.1

Type RM Length L Ch R = 1 ,23330   ,675.7,672.4,659
XS GIS Cut Line= 4
2024557.93002943191269.2506302662024135.08248176191457.182873672
2023524.30269069191772.6405679622023168.57380139191927.013482189
#Sta/Elev= 30
       0 1592.85   169.5 1567.31   442.4  1540.1     523 1527.04     597 1520.47
   663.3 1504.76   700.3 1498.68   711.3 1491.21   718.7 1487.52   733.5 1485.28
   777.8 1485.59   799.1 1490.21   850.2 1489.25   888.6 1495.27   940.4 1498.07
   995.7 1508.98  1024.2 1518.39  1073.2 1543.21  1103.5  1562.8  1128.6  1583.6
  1157.2 1587.93  1162.2 1592.38  1172.2 1606.96    1205 1628.16  1265.2 1660.87
  1347.4 1713.03  1386.6 1735.23  1451.5 1763.66  1504.8 1780.06  1537.9 1787.17
#Mann= 8 ,-1 , 0
       0      .1       0     340     .12       0     390      .1       0
  612.73     .12       0   711.3    .045       0   799.1      .1       0
 1052.73     .04       0 1160.16      .1       0
Bank Sta=711.3,799.1
XS Rating Curve= 0 ,0
Exp/Cntr(USF)=0,0
Exp/Cntr=0.3,0.1

Type RM Length L Ch R = 1 ,22658   ,933.7,943.5,955.7
XS GIS Cut Line= 4
 2024215.6248718190624.9115100152023772.64172662190893.386143453
2023168.57380139 191296.098093612022900.09916795 191544.43712954
#Sta/Elev= 30
       0 1628.32   132.2 1592.44   218.2 1570.94   320.9 1552.68   452.5 1537.58
   590.2 1525.96   639.6 1518.76   681.6  1516.5   817.1  1500.1   900.4 1495.24
   934.3 1488.77   940.3 1485.57   959.5 1485.38  1006.6 1485.51  1012.8 1488.24
    1016 1490.24  1049.1 1495.82  1069.4 1502.58    1087 1506.26  1116.8 1522.12
  1160.1 1549.98  1191.1 1562.92  1211.4 1569.04  1282.2 1580.97  1327.7 1585.94
  1359.5 1596.25  1388.5 1596.69  1403.3  1603.5  1512.5 1629.35  1609.7 1645.67
#Mann= 7 ,-1 , 0
       0      .1       0   934.3    .045       0  1012.8      .1       0
 1263.99     .04       0 1313.99      .1       0 1413.99     .04       0
 1553.99      .1       0
Bank Sta=934.3,1012.8
XS Rating Curve= 0 ,0
Exp/Cntr(USF)=0,0
Exp/Cntr=0.3,0.1

Type RM Length L Ch R = 1 ,21715   ,722.5,689.1,652
XS GIS Cut Line= 4
2024114.94688426 189873.182536392023564.57388571190108.097840648
2022913.52289962190329.5894132342022436.98042527190859.826814273
#Sta/Elev= 30
       0 1763.98      72 1747.94   109.5  1737.9   200.4  1719.8   321.7 1693.41
   410.9  1669.9   482.8 1644.51   571.4 1594.97   755.9 1503.72   772.8 1497.95
     787 1495.47   877.2 1491.78   880.6 1491.21   887.5 1485.58   970.7 1485.09
   979.7 1485.89   987.4 1491.74  1015.8 1498.68  1050.4  1515.2  1064.3 1515.73
  1074.7 1520.19  1088.5 1522.92  1329.1 1525.77  1394.1 1528.12  1433.6 1530.58
  1445.2  1532.8  1467.7  1531.8  1614.7  1537.5    1972 1544.79    1999 1546.99
#Mann= 11 ,-1 , 0
       0     .12       0     230      .1       0     400     .12       0
     550      .1       0   877.2    .045       0   987.4      .1       0
 1068.41    .035       0 1416.11     .04       0 1566.11    .035       0
 1686.11     .06       0 1866.11    .035       0
Bank Sta=877.2,987.4
XS Rating Curve= 0 ,0
Exp/Cntr(USF)=0,0
Exp/Cntr=0.3,0.1

Type RM Length L Ch R = 1 ,21025   ,595.2,549.5,500.6
XS GIS Cut Line= 4
2023604.84508072189014.0637093892023215.55686224 189376.50446453
2022832.98050959189859.7588047182022403.42109609190792.708155914
#Sta/Elev= 30
       0 1741.24    93.8  1726.8   323.1 1696.97   460.1 1671.33   514.2 1650.61
   582.1 1613.47   632.6 1578.39   653.7 1562.14   680.2 1537.65   690.9 1524.75
   730.5 1490.59   738.3 1485.68   746.9 1485.11     817 1485.11   828.2 1490.62
   854.1 1490.61   875.7 1493.94   929.1 1494.19   950.3 1498.49   964.1 1498.65
   980.4  1503.6    1029 1507.03  1237.5 1515.78  1360.3 1522.74  1562.6 1526.28
  1602.3 1528.69  1645.7    1528  1793.7 1536.28  1938.2 1536.94  2175.3 1543.78
#Mann= 10 ,-1 , 0
       0     .12       0     260      .1       0     340     .12       0
     390      .1       0   730.5    .045       0   828.2      .1       0
 1001.89    .035       0 1558.25     .06       0 1638.25    .035       0
 2108.25     .04       0
Bank Sta=730.5,828.2
XS Rating Curve= 0 ,0
Exp/Cntr(USF)=0,0
Exp/Cntr=0.3,0.1

Type RM Length L Ch R = 1 ,20476   ,533.3,484.7,436.1
XS GIS Cut Line= 4
2022873.25170461188698.6060150992022544.37027865189228.843416139
2022577.92960783190014.131718944 2022349.7261694190779.284424242
#Sta/Elev= 30
       0 1606.47    84.2 1601.81     108 1595.86   160.1 1598.15     207 1588.61
   249.5 1574.06   265.9 1580.07   288.1 1582.75   343.9 1577.17   411.6 1581.78
     556 1569.92     647 1551.74   722.5 1544.26   735.9  1537.6   761.9 1514.07
   781.11491.783   788.2 1484.94   871.3 1484.92   893.3    1490  1037.7 1493.82
  1053.9 1497.82  1349.7 1516.53  1366.1 1520.18    1399 1514.58  1445.2 1514.91
  1511.5 1517.33  1535.4 1524.95  1685.2 1526.65  1850.4 1537.65  2208.4 1541.97
#Mann= 11 ,-1 , 0
       0      .1       0     410     .12       0     470      .1       0
   781.1    .045       0   893.3      .1       0  933.95    .035       0
 1233.95      .1       0 1429.96     .06       0 1529.96     .04       0
 1639.96    .035       0 2049.96     .04       0
Bank Sta=781.1,893.3
XS Rating Curve= 0 ,0
Exp/Cntr(USF)=0,0
Exp/Cntr=0.5,0.3

Type RM Length L Ch R = 1 ,20034   ,137.6,155.8,148.8
XS GIS Cut Line= 4
2022328.93119683188826.5067849312022146.73177908189593.713059518
2022496.03368726190002.3822089882022305.80573293190759.432738659
#Sta/Elev= 30
       01531.444  86.4651527.755  99.9541521.483 113.4421525.103     1911515.489
  207.861509.875 238.209 1511.45 265.1861503.475  271.931506.749 342.7441504.082
 373.0921508.426  450.651503.229  514.72 1506.98 565.301 1503.35 629.3711508.695
 706.9281494.364 737.2771493.054 788.5441501.618 827.5561490.397 973.9921485.023
1016.4121483.994 1062.021485.0251135.5761491.3021163.1551502.0291266.7391513.843
1360.7721515.6081384.452 1522.681580.6551525.3751773.4761536.8612106.7371540.444
#Mann= 18 ,-1 , 0
       0     .04       0     230     .06       0     330      .1       0
     400     .06       0     430     .04       0     530      .1       0
     630     .04       0     740      .1       0  848.54     .04       0
  928.54      .1       0 973.992    .045       0 1062.02      .1       0
 1356.15     .08       0 1456.15     .04       0 1566.15    .035       0
 1966.15     .04       0 1986.15     .06       0 2066.15     .08       0
#XS Ineff= 2 , 0
          913.17 1522.36 1137.72         1521.57
Permanent Ineff=
       F       F
Bank Sta=973.992,1062.02
XS Rating Curve= 0 ,0
Exp/Cntr(USF)=0,0
Exp/Cntr=0.5,0.3

Type RM Length L Ch R = 1 ,19835   ,243.8,239.1,233.9
XS GIS Cut Line= 4
2022167.04932373188784.7990004542021970.16856064 189617.73917272
2022366.49752638 190159.388759242022256.40614702190775.900483735
#Sta/Elev= 30
       01566.875 200.0971570.109 260.7791567.195 270.8931564.294 348.4311567.997
 378.7721563.487 446.1971565.238 469.7961561.193 483.2811562.634 500.1371558.467
 520.3641559.985 540.592 1555.99  618.131569.328 756.3511578.672 790.0631571.084
 854.1171536.065 894.4051498.199 910.6661489.0281065.148 1490.45 1194.22 1484.76
1203.3741483.781 1288.741484.7491325.4451489.1831341.5891499.681 1418.831518.587
1455.4181522.8471631.6311524.9471811.5991535.0022018.228 1535.59 2153.321539.695
#Mann= 13 ,-1 , 0
       0      .1       0     470     .04       0     560      .1       0
  975.89     .04       0 1005.89      .1       0 1145.89     .04       0
 1194.22    .045       0 1288.74      .1       0 1315.89     .04       0
 1365.89      .1       0 1495.89    .035       0 1997.06     .06       0
 2097.06     .08       0
#XS Ineff= 2 , 0
         1163.01 1523.15 1320.96         1523.15
Permanent Ineff=
       F       F
Bank Sta=1194.22,1288.74
XS Rating Curve= 0 ,0
Exp/Cntr(USF)=0,0
Exp/Cntr=0.5,0.3

Type RM Length L Ch R = 1 ,19596   ,453.4,409.2,388.6
XS GIS Cut Line= 4
2021447.09297381188975.9523927992021746.54152571189706.959151843
2022195.71435356190310.2599108132022266.17283636190741.818117959
#Sta/Elev= 30
       0 1833.96    85.7 1815.13   156.3 1792.53   237.9 1784.13   429.3 1742.09
   528.6 1734.76     603 1721.75   666.9  1715.8   696.9 1710.09   732.1 1690.63
   787.4 1653.69   843.8 1601.36   902.5 1552.52   950.6 1501.28     967 1487.37
   984.5 1484.74    1012 1487.41  1040.6 1483.68    1085 1487.74  1110.1 1481.54
  1167.4 1485.38  1228.4 1484.55  1271.8 1482.11  1293.8 1484.87  1308.1 1496.28
  1351.5 1501.72  1416.9 1521.09  1543.4 1523.42  1719.6 1532.24  1979.4 1538.55
#Mann= 6 ,-1 , 0
       0      .1       0  1228.4    .045       0  1293.8      .1       0
 1449.96    .035       0 1862.11     .06       0 1962.11     .08       0
Bank Sta=1228.4,1293.8
XS Rating Curve= 0 ,0
Exp/Cntr(USF)=0,0
Exp/Cntr=0.3,0.1

Type RM Length L Ch R = 1 ,19187   ,469.8,459.2,454.3
XS GIS Cut Line= 4
2021130.02980122189539.6202551942021477.91856004190063.655221015
2021944.70600859190548.0572902612022204.52166391190812.276600759
#Sta/Elev= 30
       0 1963.68   128.2  1871.4   225.6 1811.21   268.9  1781.9   314.5  1757.2
   359.3 1737.34   422.5 1698.41   454.5 1676.09   515.7 1627.25   541.8 1611.09
   591.8  1574.2   619.9 1558.71   731.8  1513.2   759.1 1493.06  768.731488.422
   777.8 1481.83     783 1480.77   816.1 1482.18   868.2 1479.63   926.3 1480.23
   936.8 1485.67   961.91488.425  1088.7 1497.69  1202.4 1513.32  1278.5 1519.26
  1401.4 1520.07  1559.7 1531.93  1622.4 1532.79  1641.8 1536.42  1672.3 1538.03
#Mann= 8 ,-1 , 0
       0      .1       0  768.73    .045       0   961.9      .1       0
    1019    .035       0 1411.71     .06       0 1441.71     .08       0
 1541.71     .06       0 1581.71     .08       0
Bank Sta=768.73,961.9
XS Rating Curve= 0 ,0
Exp/Cntr(USF)=0,0
Exp/Cntr=0.3,0.1

Type RM Length L Ch R = 1 ,18728   ,459.4,458.3,456
XS GIS Cut Line= 4
2020812.96662862 190024.022324442021138.83711157190398.333014312
2021579.20262906190799.0656352342021852.22924991191129.339773356
#Sta/Elev= 30
       0 1870.12    53.2  1838.4   109.1 1809.69   131.2 1794.98   427.6 1572.86
   457.9  1553.8   481.1 1543.13   504.9 1534.76   529.9 1528.29   581.8 1519.24
   641.4 1506.13   673.4 1494.98   691.2 1491.73   701.8 1486.11   722.2 1479.19
   734.3    1479   806.3 1479.28     811 1480.51   819.8 1486.06   859.7 1488.81
   950.3 1489.48   973.5 1494.01  1010.8 1506.92    1040  1514.7  1094.3 1521.49
  1216.9 1532.05  1280.7  1540.4    1353 1553.72    1485 1584.62  1520.2 1589.49
#Mann= 3 ,-1 , 0
       0      .1       0   701.8    .045       0   819.8      .1       0
Bank Sta=701.8,819.8
XS Rating Curve= 0 ,0
Exp/Cntr(USF)=0,0
Exp/Cntr=0.3,0.1

Type RM Length L Ch R = 1 ,18270   ,576,577.9,578.1
XS GIS Cut Line= 4
2020513.51807672190442.3695660622020852.59952519190759.432738659
2021319.38697374191164.5690147562021548.37704284191384.751773504
#Sta/Elev= 30
       0 1800.04    47.3 1771.93    96.7 1738.69   119.2 1730.42   154.3 1711.91
     236 1662.16   312.3    1609   370.6 1563.62   408.9 1541.26     443 1529.61
   473.7 1522.56   638.8 1495.79   661.1 1484.34   686.9 1479.07   703.9 1478.78
   756.5 1479.36   773.4 1485.85   935.6 1487.25   947.2 1491.49   963.5 1501.58
   977.6 1511.93   986.3 1522.25  1012.2 1536.29  1100.1 1575.82    1154 1596.36
  1252.7 1618.21  1281.6 1616.27  1293.2 1623.18  1304.8 1625.25    1400 1630.29
#Mann= 6 ,-1 , 0
       0      .1       0   661.1    .045       0   773.4      .1       0
 1152.31     .04       0 1272.31     .06       0 1292.31    .035       0
Bank Sta=661.1,773.4
XS Rating Curve= 0 ,0
Exp/Cntr(USF)=0,0
Exp/Cntr=0.3,0.1

Type RM Length L Ch R = 1 ,17692   ,607.8,593.3,577.8
XS GIS Cut Line= 4
2020029.11600748190856.3131525082020539.94000777 191239.43115273
2020914.25069764191560.8979805022021297.36869787191776.677084076
#Sta/Elev= 30
       0 1916.97    51.9 1886.49   111.5 1844.72   150.3    1823   183.1 1797.71
   248.7 1735.67   332.9 1664.23   452.6  1572.8   518.2 1533.78     551 1519.92
   584.8 1511.66   709.8 1494.75   791.3 1489.45   822.2 1482.34   848.2 1477.32
   891.4 1477.22     903  1479.6   912.3 1477.12   933.2 1477.11     939  1477.4
   947.6 1481.54    1003 1487.54  1047.2 1507.29  1060.1 1510.41  1246.6 1525.53
  1327.1 1537.96  1385.7 1543.37  1419.6 1549.43  1513.7 1572.34  1571.6 1578.32
#Mann= 3 ,-1 , 0
       0      .1       0   822.2    .045       0   947.6      .1       0
#XS Ineff= 2 , 0
          751.86 1530.26
Permanent Ineff=
       F       F
Bank Sta=822.2,947.6
XS Rating Curve= 0 ,0
Exp/Cntr(USF)=0,0
Exp/Cntr=0.3,0.1

Type RM Length L Ch R = 1 ,17098   ,681.1,628.5,571.9
XS GIS Cut Line= 4
2019769.30035215191477.2285321782020156.82200755191732.640532326
2020473.88518015191930.8050151992021328.19428409192128.969498073
#Sta/Elev= 30
       0 1892.07    39.9 1894.74      80 1894.58   107.5 1888.74   127.2 1880.03
   162.6 1854.46   227.5 1800.48   252.9 1775.75   266.5 1764.99   288.3 1743.09
   331.7 1706.16     350 1693.05   394.4 1656.75   429.7 1624.17   449.4 1608.95
     481 1579.29     585 1506.98   612.7 1492.08  631.191485.626   650.1 1481.46
   658.5 1477.11   747.7 1476.94   754.8 1478.09   766.7 1485.04  785.511485.626
  1018.6  1493.5  1075.8 1497.16  1170.1  1506.7  1624.8 1528.43    1715 1536.25
#Mann= 6 ,-1 , 0
       0      .1       0  631.19    .045       0  785.51      .1       0
  834.12    .035       0  938.02      .1       0 1038.02    .035       0
#XS Ineff= 2 , 0
                          930.95            1525
Permanent Ineff=
       F       F
Bank Sta=631.19,785.51
XS Rating Curve= 0 ,0
Exp/Cntr(USF)=0,0
Exp/Cntr=0.3,0.1

Type RM Length L Ch R = 1 ,16470   ,602.4,600.6,594.1
XS GIS Cut Line= 4
 2019778.1076625 192446.032670672020037.92331783192476.858256895
2020760.12276652 192401.996118922021588.00993941192234.657222272
#Sta/Elev= 30
       0 1597.96   322.6  1569.3   346.8  1562.5   385.3 1541.24   421.5 1512.93
   441.4 1492.01  446.021484.384   451.3 1477.68   507.3 1476.96     537 1477.08
   540.3 1477.72  546.871484.386   566.7 1486.02   629.4 1484.62   764.6 1486.14
   808.1 1490.84   899.9 1493.59  1025.7 1503.27  1120.1 1507.85  1363.8 1513.69
  1417.4 1516.69  1443.1 1521.78  1521.1 1519.49  1544.6 1523.23    1599 1527.06
  1668.6 1537.63  1682.5 1538.13  1772.2 1556.61  1798.9 1564.21  1832.3 1566.47
#Mann= 7 ,-1 , 0
       0      .1       0  446.02    .045       0  546.87      .1       0
  601.64    .035       0  691.64      .1       0  891.64    .035       0
 1797.71     .04       0
#XS Ineff= 2 , 0
                          799.43         1504.21
Permanent Ineff=
       F       F
Bank Sta=446.02,546.87
XS Rating Curve= 0 ,0
Exp/Cntr(USF)=0,0
Exp/Cntr=0.3,0.1

Type RM Length L Ch R = 1 ,15869   ,359.8,362.3,370.4
XS GIS Cut Line= 4
2019769.30035215192714.6556363432020280.12435245193053.737084815
2020896.63607694192904.0128088662021737.73421536192710.251981168
#Sta/Elev= 30
       0 1529.61   107.8 1521.33   222.6 1517.77   359.5 1514.91   501.6 1515.87
     600 1512.91   686.3 1509.87   709.9 1502.46   733.5 1489.96   747.1 1486.96
   757.2 1482.08   784.2 1480.47   814.6 1476.45   899.7 1475.85   932.7 1480.38
   990.1 1482.25  1064.4 1496.06  1142.1 1500.61    1442  1512.5  1556.3  1513.2
  1596.9  1517.1  1723.5  1522.3  1802.2 1527.88  1899.9 1529.39  1930.2 1533.52
  2024.5 1538.93  2044.7  1541.6  2064.9 1547.22  2088.4 1547.45  2110.7 1550.68
#Mann= 7 ,-1 , 0
       0      .1       0     600    .035       0  703.12      .1       0
   784.2    .045       0   932.7      .1       0 1213.12    .035       0
 1777.55     .06       0
Bank Sta=784.2,932.7
XS Rating Curve= 0 ,0
Exp/Cntr(USF)=0,0
Exp/Cntr=0.3,0.1

Type RM Length L Ch R = 1 ,15507   ,727.4,778.8,846.1
XS GIS Cut Line= 4
2020103.48885043193150.6174986642020381.40842147193357.589291887
2021028.74573219193300.3417746132021891.86214649193216.672326289
#Sta/Elev= 30
       0 1504.11   124.4    1504   228.8 1509.19   288.8 1508.35   344.1 1504.37
   411.7 1496.05   434.5 1490.77   484.2 1482.98   520.4 1482.15   543.5 1479.07
   569.8 1478.47     583 1474.86   599.5 1474.68   652.2 1474.87     662 1478.59
   737.6 1487.86   823.4 1494.62  1014.5 1503.63  1060.3 1504.42  1248.5 1515.29
  1377.1 1519.61  1413.3 1522.29  1466.6 1522.99  1485.8 1527.07  1518.8 1530.27
  1657.2 1536.11  1729.8 1545.78  1749.5 1546.66  1808.9 1557.36  1863.5 1569.36
#Mann= 13 ,-1 , 0
       0     .05       0      50      .1       0      90     .05       0
     210    .035       0     220     .05       0  436.52      .1       0
  536.52     .12       0   569.8    .045       0     662     .12       0
  736.52      .1       0  826.52    .035       0 1716.38     .06       0
 1816.38      .1       0
Bank Sta=569.8,662
XS Rating Curve= 0 ,0
Exp/Cntr(USF)=0,0
Exp/Cntr=0.3,0.1

Type RM Length L Ch R = 1 ,14728   ,733.1,775.6,833.8
XS GIS Cut Line= 4
2020103.48885043193234.286946988 2020359.3901456 193714.28536106
2020566.36193882194167.8618440812020601.59118022194480.521361503
#Sta/Elev= 30
       0 1504.37   164.1 1509.03   345.9 1498.84   583.1 1495.75   621.6 1492.34
   651.3 1481.89   687.6 1475.35   720.1 1476.19   745.3 1480.44     790 1479.65
     803 1476.25   828.3 1475.15   842.7 1471.33   860.7 1471.15   882.4 1471.52
   891.1 1475.54   906.4 1477.31   913.8 1482.11   924.3 1491.84   950.9 1523.33
   968.9 1538.92     993 1555.69    1023 1571.86  1054.3 1580.59  1097.3 1587.69
  1131.6 1587.75  1209.6 1578.38  1239.3 1564.45  1328.4 1576.93  1357.2 1578.21
#Mann= 8 ,-1 , 0
       0      .1       0     150     .05       0     280      .1       0
     390     .05       0     500      .1       0   828.3    .045       0
   891.1      .1       0 1342.52     .04       0
Bank Sta=828.3,891.1
XS Rating Curve= 0 ,0
Exp/Cntr(USF)=0,0
Exp/Cntr=0.3,0.1

Type RM Length L Ch R = 1 ,13953   ,393.5,390.6,389.6
XS GIS Cut Line= 4
2020069.72749409193227.9261117362020074.62044428193438.322970095
2019722.32803029193873.7955373972019511.93117193194133.121897701
#Sta/Elev= 30
       0 1506.16    88.9 1507.21   184.1 1502.36   238.4 1496.53   272.6 1486.32
   298.9 1481.36   383.3 1476.04   424.3  1470.8   433.6 1471.44   446.6 1467.79
   463.5 1470.24   480.1 1470.43     493 1467.45   517.6 1466.93   547.7 1467.28
   558.4 1470.07   568.8 1473.61   579.2 1474.85   589.7 1481.32   594.9 1485.99
   605.3  1498.9   624.9 1520.81   662.7 1551.97   720.9 1594.57   750.8 1611.82
   771.8 1621.82   811.5 1631.21     856 1635.21  1058.8 1642.41  1104.5  1641.1
#Mann= 5 ,-1 , 0
       0     .05       0      80      .1       0   480.1    .045       0
   558.4      .1       0  850.58    .035       0
Bank Sta=480.1,558.4
XS Rating Curve= 0 ,0
Exp/Cntr(USF)=0,0
Exp/Cntr=0.3,0.1

Type RM Length L Ch R = 1 ,13562   ,453.9,467.5,469.5
XS GIS Cut Line= 4
 2019976.7614404193081.1376059042019864.22358593193134.960058042
2019511.93117193  193521.50312342019286.85546299193815.080135064
#Sta/Elev= 30
       0 1505.38    41.1 1503.19    92.7 1498.49   126.6 1497.74     147 1495.91
   179.9 1490.34   233.9 1474.32   244.4 1472.76   263.9 1471.72   286.4 1472.43
   302.8 1469.84     343 1469.24     357 1468.07     371 1465.85   458.7 1465.79
   472.9 1466.05   477.7    1468     494 1474.63   507.9 1475.81   530.6 1491.48
     566 1506.13   603.1 1525.05   648.7 1546.64   666.8 1553.17   699.8 1563.09
     762 1576.99   876.6 1595.72   918.4  1598.1   950.7 1601.14  1017.7 1602.06
#Mann= 4 ,-1 , 0
       0     .05       0      10      .1       0     357    .045       0
   477.7      .1       0
Bank Sta=357,477.7
XS Rating Curve= 0 ,0
Exp/Cntr(USF)=0,0
Exp/Cntr=0.3,0.1

Type RM Length L Ch R = 1 ,13095   ,492.1,487.9,481
XS GIS Cut Line= 4
2019650.08150643192726.912174546 2019565.5119969192823.563042584
2019239.31531727193337.0207790332019106.42037372193669.258137913
#Sta/Elev= 30
       0 1522.06   116.8 1502.13   211.4  1491.6   223.2 1487.97   238.6 1474.88
   256.4 1465.33   263.6 1462.19   287.3 1461.51   311.1 1464.24   382.4  1467.5
   396.7 1466.25   415.7 1470.41     429 1469.53   443.6 1473.49   458.5 1470.59
   468.1 1473.17   526.2 1476.06   551.2 1479.14     566 1482.77   576.7 1486.99
   591.6 1487.78   601.1 1493.99   623.4 1503.69   658.1 1516.69     689 1526.04
   724.4 1533.94   789.2 1543.16   933.4 1552.45    1033 1554.86  1094.6    1560
#Mann= 3 ,-1 , 0
       0      .1       0   256.4    .045       0   311.1      .1       0
Bank Sta=256.4,311.1
XS Rating Curve= 0 ,0
Exp/Cntr(USF)=0,0
Exp/Cntr=0.3,0.1

Type RM Length L Ch R = 1 ,12607   ,656.3,648.3,635
XS GIS Cut Line= 4
2019354.08822306192279.9019098722019148.70512848192551.732476228
2018913.11863764192998.7427409022018701.69486381193512.200477352
#Sta/Elev= 30
       0 1733.57      82 1671.87   163.7 1616.31   175.9 1603.48   189.3 1599.92
   238.7 1565.26     251 1554.71   263.4 1551.03   296.2 1529.49   316.8 1519.06
   393.4 1491.57   408.2 1483.91   419.3 1472.32   426.7  1467.8   441.5 1463.06
   452.7 1460.08     512 1459.94   526.9 1460.25     539 1464.14   580.3 1466.86
   593.6 1470.87   604.7 1469.44   916.7 1510.51  1012.5 1518.42  1108.3  1533.8
  1143.8 1534.15  1200.6 1543.04  1230.9 1551.28  1324.8  1562.1  1401.3 1574.38
#Mann= 8 ,-1 , 0
       0      .1       0     280     .12       0   441.5    .045       0
     539      .1       0  905.99    .035       0 1045.99      .1       0
 1165.99    .035       0 1255.99      .1       0
Bank Sta=441.5,539
XS Rating Curve= 0 ,0
Exp/Cntr(USF)=0,0
Exp/Cntr=0.3,0.1

Type RM Length L Ch R = 1 ,11959   ,794.1,770.6,733.5
XS GIS Cut Line= 4
2018623.16603353192032.2340605262018556.71856175 192249.69851361
2018357.37614643192811.4816840792018309.05071241193312.858062024
#Sta/Elev= 30
       0  1626.7    97.9  1611.7   159.8 1604.21   193.9 1598.09   204.2 1594.24
     218 1586.82   233.3 1574.63   256.1 1548.02   274.4 1533.73     284  1524.2
   292.4 1513.89   304.8  1493.5   311.8 1484.88   336.2 1463.11   346.6 1459.51
   357.1 1457.12   392.6 1456.59   419.7 1458.96   467.1 1463.14   492.8 1461.28
   517.2 1466.83   541.5 1470.18     611 1476.36   654.7 1485.03   680.8  1484.3
   691.3 1489.52    1056 1518.52    1140 1533.87  1281.7 1551.48  1327.2 1558.77
#Mann= 3 ,-1 , 0
       0      .1       0   346.6    .045       0   419.7      .1       0
Bank Sta=346.6,419.7
XS Rating Curve= 0 ,0
Exp/Cntr(USF)=0,0
Exp/Cntr=0.3,0.1

Type RM Length L Ch R = 1 ,11188   ,651,793.8,928
XS GIS Cut Line= 4
 2018296.9693539192026.1933812732017741.22686269192183.251041834
2017753.30822119192654.4240235182017439.19290007 193071.23089193
#Sta/Elev= 30
       0    1540    59.1 1530.47   159.8 1517.33   170.8 1517.87   381.4 1505.12
   490.5 1501.97   577.4  1497.2   651.4 1498.47   664.5 1494.34   677.6 1476.35
     694 1461.77   703.9 1457.74   723.6 1453.72   766.4 1453.31   782.6 1453.76
   795.8 1457.17   864.7 1464.82   890.9 1464.71   900.8 1469.72  1005.8 1486.05
  1018.9 1489.92  1118.2    1509  1159.1 1518.31  1278.5 1549.16    1323 1562.62
  1387.7 1585.69    1487 1628.44    1513  1635.8  1537.3 1640.53  1570.8 1643.95
#Mann= 3 ,-1 , 0
       0      .1       0   703.9    .045       0   795.8      .1       0
Bank Sta=703.9,795.8
XS Rating Curve= 0 ,0
Exp/Cntr(USF)=0,0
Exp/Cntr=0.3,0.1

Type RM Length L Ch R = 1 ,10394   ,980.2,1081.2,1153.7
XS GIS Cut Line= 4
2018339.25410867191941.623871741 2017511.6810511 192044.31541903
2016998.22331465 191965.78658875 2016611.6198425191814.769607441
#Sta/Elev= 30
       0 1542.19    28.9 1532.14    45.5 1532.43   128.1 1518.29   230.6 1506.25
   481.9 1497.75   690.1 1482.91   882.1 1478.64   938.5 1472.81   978.3 1464.06
  1071.3 1460.66  1109.3 1455.64  1138.1 1453.32  1181.3 1455.54  1200.7 1458.74
    1204  1463.1  1221.6 1500.34  1253.8 1526.08  1353.4 1593.23  1367.5 1609.31
  1395.6 1635.83  1430.9 1661.51  1480.5 1704.85  1501.3 1718.31  1564.7 1780.98
  1637.6 1837.01  1666.8  1866.7  1716.3 1909.97  1738.9  1921.4  1768.4  1926.4
#Mann= 3 ,-1 , 0
       0      .1       0  1109.3    .045       0  1181.3      .1       0
Bank Sta=1109.3,1181.3
XS Rating Curve= 0 ,0
Exp/Cntr(USF)=0,0
Exp/Cntr=0.3,0.1

Type RM Length L Ch R = 1 ,9313    ,542.3,524.3,490.7
XS GIS Cut Line= 4
2018200.31848587191893.2984377222018049.30150456191778.525531927
2017898.28452325191210.7016822062017300.25727727 190860.34228557
#Sta/Elev= 30
       0 1511.61   136.2  1497.3   154.1  1492.9   179.2 1492.66   230.9 1482.51
     258 1481.03   302.2 1470.06   342.9 1463.86   397.5 1457.63   482.1 1453.28
   526.2 1447.38   526.2 1447.37   534.3 1445.18     567 1444.94   611.1 1445.22
   617.9 1446.99   628.1 1452.13   631.5 1456.12   648.5 1460.04   668.8  1488.9
   682.4 1501.65   709.6 1507.93     783 1514.67   862.1 1529.68   972.4 1546.51
  1033.3 1558.91  1109.4 1578.24  1266.5  1626.2  1336.9 1654.83  1470.3 1716.48
#Mann= 3 ,-1 , 0
       0      .1       0   526.2    .045       0   617.9      .1       0
Bank Sta=526.2,617.9
XS Rating Curve= 0 ,0
Exp/Cntr(USF)=0,0
Exp/Cntr=0.3,0.1

Type RM Length L Ch R = 1 ,8789    ,810.9,762.2,677.5
XS GIS Cut Line= 4
2018701.69486381191699.9967016462018580.88127876191476.491569309
2018151.99305185190969.074512112 2017396.9081453190642.877832485
#Sta/Elev= 30
       0 1613.38    26.9 1605.07      64 1590.47   187.2 1537.82   275.9 1509.85
   348.9 1481.41     353 1478.83   362.8 1463.94   383.8 1453.33   401.8 1447.81
   426.2 1443.81   471.7 1444.18   499.3 1447.84   560.2 1448.16   576.6 1448.98
   593.8  1452.7   620.7 1453.51   653.9 1458.08   667.2 1461.78     684 1462.29
   706.8 1470.09   755.7 1478.82   985.2 1499.38  1235.6 1515.63  1310.2 1525.78
  1346.2 1532.44  1410.5 1547.93  1553.5  1587.3  1689.3 1629.97    1741  1651.2
#Mann= 3 ,-1 , 0
       0      .1       0   401.8    .045       0   499.3      .1       0
Bank Sta=401.8,499.3
XS Rating Curve= 0 ,0
Exp/Cntr(USF)=0,0
Exp/Cntr=0.3,0.1

Type RM Length L Ch R = 1 ,8027    ,775.6,745,697.4
XS GIS Cut Line= 4
2019257.43735503190697.2439457562018997.68814718190691.203266504
2018339.25410867190727.4473420182017469.39629633190576.430360709
#Sta/Elev= 30
       0 1770.17    21.7 1751.09    70.9 1716.82   235.4 1608.11   333.6 1534.85
   356.6  1513.3   363.1 1502.56     373 1492.37   382.9 1479.18   402.6 1449.86
   415.7 1442.35   461.7 1441.06   471.6 1442.15   497.9 1442.21   540.6 1447.03
   563.6 1445.02     580 1447.54   629.3 1447.24   704.9  1454.9   780.4  1470.6
   796.9 1470.54   816.6 1475.56   933.9 1484.45  1191.5 1498.62  1384.6 1514.53
  1524.5 1540.45  1584.4 1557.17    1611 1561.66  1752.1 1603.86  1802.1 1621.06
#Mann= 7 ,-1 , 0
       0      .1       0     180     .12       0  269.82      .1       0
   415.7    .045       0   471.6      .1       0  769.82     .05       0
 1059.25      .1       0
Bank Sta=415.7,471.6
XS Rating Curve= 0 ,0
Exp/Cntr(USF)=0,0
Exp/Cntr=0.3,0.1

Type RM Length L Ch R = 1 ,7282    ,1038.5,1047.9,1031.9
XS GIS Cut Line= 4
2018955.40339241189736.7759446332018629.20671278 189936.11835996
2018145.95237259 190244.193001832017469.39629633190503.942209681
#Sta/Elev= 30
       0 1864.69    48.3 1837.78   155.9 1768.94   202.2 1731.26   267.4 1681.18
   305.9 1653.47   336.6 1628.28   363.6 1609.42   417.8 1565.01   429.5 1557.32
   464.4 1529.68   488.7 1513.45   530.6 1477.06   557.9 1444.91   561.8 1442.02
   569.6 1439.76   592.7 1436.06   662.9 1436.18   685.4  1440.5   779.7 1445.06
   865.3 1459.59   950.8 1482.08   968.9 1479.13   981.7 1483.81   996.9 1485.31
  1197.3 1496.75    1289 1510.36  1432.8 1546.07  1546.1 1577.48  1680.1 1623.94
#Mann= 3 ,-1 , 0
       0      .1       0   569.6    .045       0   685.4      .1       0
Bank Sta=569.6,685.4
XS Rating Curve= 0 ,0
Exp/Cntr(USF)=0,0
Exp/Cntr=0.3,0.1

Type RM Length L Ch R = 1 ,6234    ,760.7,751.5,745.4
XS GIS Cut Line= 4
2018454.02701446188897.1215285562017952.65063652189174.992774164
2017408.98950381189573.6776048192017106.95554119189827.386133418
#Sta/Elev= 30
       0 1597.45    47.8 1573.08      74 1562.29   175.3 1535.97   426.8 1493.46
   523.4 1484.75   565.4 1476.35   629.8 1456.46   684.3 1445.58   715.3 1441.28
   758.7  1439.8   794.3 1434.53   883.9 1432.18   908.4  1435.1   947.2 1437.43
   959.4 1441.97  1020.4 1454.03  1040.8 1463.16    1057 1474.81  1071.6 1476.86
  1226.5 1586.22  1338.3 1647.84  1402.5 1687.51    1434 1702.04  1445.4  1710.7
  1450.9 1724.22  1454.9 1731.21  1475.4 1741.45  1539.7 1762.09  1641.9 1777.14
#Mann= 3 ,-1 , 0
       0      .1       0   794.3    .045       0   908.4      .1       0
Bank Sta=794.3,908.4
XS Rating Curve= 0 ,0
Exp/Cntr(USF)=0,0
Exp/Cntr=0.3,0.1

Type RM Length L Ch R = 1 ,5482    ,568,571.1,575.4
XS GIS Cut Line= 4
2017886.20316474188268.8908863122017469.39629633188564.884169677
2016961.97923913189023.9757928552016720.35206904189229.358887435
#Sta/Elev= 30
       0 1560.17   143.5 1515.21     243 1497.74   360.6 1486.15   591.3 1472.52
   601.8 1469.02   624.6 1455.63   655.2  1434.4   692.4 1429.15   724.9 1432.14
     738 1429.81     775 1433.61   806.2 1431.89   817.8 1429.35   841.4 1429.25
   887.5 1431.92   901.5 1435.42   925.4 1451.54   947.5  1462.1   987.4 1476.02
  1002.1 1486.95  1022.8 1489.23  1036.3 1500.17  1119.5 1540.23  1208.2    1590
  1350.3 1660.76    1370  1664.4  1423.5 1661.26  1470.9 1653.63  1512.6 1642.85
#Mann= 3 ,-1 , 0
       0      .1       0   806.2    .045       0   887.5      .1       0
Bank Sta=806.2,887.5
XS Rating Curve= 0 ,0
Exp/Cntr(USF)=0,0
Exp/Cntr=0.3,0.1
